HEC-RAS study MFRFBUCKRV.prj: MFRFBUCKRV

--- MFRFBUCKRV.g01 (geometry) --- (continued)

Type RM Length L Ch R = 1 ,8884    ,408.3,408.8,408.4
XS GIS Cut Line= 2
2188366.93402289630003.8857287082188810.48302843630443.933031571
#Sta/Elev= 30
       0 2125.71    24.4  2116.5    32.9  2115.5    47.3  2111.5      64 2104.16
    69.4 2101.29    89.5 2084.75   109.3 2071.61   120.6 2062.25   131.3 2055.51
   143.8 2050.97   160.2 2049.55   176.4 2051.84   219.6 2051.99   253.5  2056.3
   268.8 2055.96   291.5 2053.14   351.1 2055.02   384.9 2054.46   456.2 2055.94
   468.5 2052.39   482.6  2052.4   490.3 2055.91   501.6 2064.71   519.4 2083.26
   524.3 2086.79     542 2088.27   553.3 2095.04   584.5  2101.2   624.8 2111.53
#Mann= 4 ,-1,0
       0      .1       0   468.5    .045       0   482.6      .1       0
     520     .06       0
#XS Ineff= 2 , 0
          353.19 2071.93
Permanent Ineff=
       F       F
Bank Sta=468.5,482.6
XS Rating Curve= 0 ,0
Exp/Cntr(USF)=0,0
Exp/Cntr=0.3,0.1

Type RM Length L Ch R = 1 ,8475    ,207.8,207.8,205
XS GIS Cut Line= 2
 2188200.0195287 630139.284898822188564.19660693630585.168372809
#Sta/Elev= 30
       0 2126.84    25.5  2116.3    38.2 2108.58    50.8 2102.98    58.3 2097.67
    76.1    2088    95.1 2073.87   141.9 2044.02   152.2 2042.56   183.6  2042.9
   191.9 2042.09   198.7 2041.56   207.92042.064   219.4    2045   245.2 2042.78
   255.5 2043.44   276.2 2041.61   296.8 2046.29   314.2 2044.57   327.8 2045.74
   334.1 2047.63   353.6 2056.96   374.3 2062.03   420.8 2066.33   449.2 2066.53
   480.8  2068.8   503.4 2073.34   529.2 2073.62   541.6 2079.29   575.7 2089.81
#Mann= 4 ,-1,0
       0      .1       0   191.9    .045       0   207.9      .1       0
     500     .06       0
#XS Ineff= 2 , 0
          143.17 2054.25  293.99         2059.53
Permanent Ineff=
       F       F
Bank Sta=191.9,207.9
XS Rating Curve= 0 ,0
Exp/Cntr(USF)=0,0
Exp/Cntr=0.3,0.1

Type RM Length L Ch R = 1 ,8267    ,113.8,113.3,113.5
XS GIS Cut Line= 4
2188054.11525056630243.1687448542188114.81143026630350.554293563
2188217.52804207630460.2743107232188552.52426468630584.001138584
#Sta/Elev= 30
       0 2108.52    61.1 2067.15      85 2054.51    89.6 2051.37   112.6 2045.46
   126.9 2037.55   151.6 2036.34   171.5 2033.28   179.9 2032.53   192.7 2033.25
   201.4 2034.59   213.9 2035.04   231.1 2037.79   269.4 2039.92   273.3 2040.74
   282.6 2044.34   306.3 2046.61   323.1 2049.87   344.9 2051.25   379.2 2055.17
   404.4  2060.9   421.4 2063.58   441.5 2064.67   472.6    2065   488.2 2067.19
   519.5 2069.67   531.8 2071.69   575.4 2073.52   587.7 2078.09   630.8 2087.21
#Mann= 4 ,-1,0
       0      .1       0   171.5    .045       0   192.7      .1       0
  463.65     .06       0
Bank Sta=171.5,192.7
XS Rating Curve= 0 ,0
Exp/Cntr(USF)=0,0
Exp/Cntr=0.3,0.1

Type RM Length L Ch R = 1 ,8154    ,227.8,234.8,235.4
XS GIS Cut Line= 4
2187954.90034143 630313.202798362188007.42588155630401.912599467
2188143.99228589630534.9773011292188446.30595019630637.693912938
#Sta/Elev= 30
       0 2100.93    18.6 2086.36    32.5 2084.35      36  2082.3    47.6    2074
    56.4 2065.75    65.1 2061.96    88.5  2045.9   109.7 2037.92   132.1 2034.59
   148.8 2035.21   162.32030.882     171 2029.87   181.52030.894   210.9 2032.81
   243.8 2028.92   254.9 2029.79   268.3 2033.75     287 2034.77   302.4 2039.96
   315.1  2041.8   336.2 2047.52   365.8 2048.69   399.7 2054.95   443.8 2060.09
   481.7 2061.59   499.6 2066.01     539 2072.92     577 2078.68   613.1 2081.83
#Mann= 5 ,-1,0
       0      .1       0   162.3    .045       0   181.5      .1       0
  393.77     .06       0  573.77      .1       0
#XS Ineff= 2 , 0
                          257.56          2044.7
Permanent Ineff=
       F       F
Bank Sta=162.3,181.5
XS Rating Curve= 0 ,0
Exp/Cntr(USF)=0,0
Exp/Cntr=0.3,0.1

Type RM Length L Ch R = 1 ,7919    ,188.6,198.8,205.2
XS GIS Cut Line= 2
2187863.85607187630352.8887620132188136.98888054630826.785857405
#Sta/Elev= 30
       0  2096.6    32.7 2081.87    50.2 2075.92    64.7 2072.14    92.7 2062.47
   104.8 2056.66   112.8  2054.5   123.5 2053.15   143.5 2045.36   157.3  2043.8
     182  2038.4   202.5 2037.06   216.9 2033.06   249.6 2030.22   281.6 2031.58
   314.3 2030.92   321.1 2029.39   331.4 2022.64   335.82021.403     342 2020.93
   356.8 2021.39   361.1 2022.26   369.5 2027.18   378.3 2034.93   388.1 2045.97
     390 2046.52   406.6 2047.12   415.8 2051.78   448.2 2059.92     547 2076.13
#Mann= 5 ,-1,0
       0      .1       0   335.8    .045       0   356.8      .1       0
     360     .06       0     540      .1       0
Bank Sta=335.8,356.8
XS Rating Curve= 0 ,0
Exp/Cntr(USF)=0,0
Exp/Cntr=0.3,0.1

Type RM Length L Ch R = 1 ,7720    ,235.3,229,218.8
XS GIS Cut Line= 4
2187797.32372104630394.9091941172187872.02671144630520.970490428
2187792.65478414630820.9496862792187862.68883764630954.014387941
#Sta/Elev= 30
       0 2091.33    13.4    2084    44.5 2069.46    84.1 2052.86   129.3 2040.69
   146.7 2034.81     155 2032.74   171.6 2028.72   204.7 2023.29     213 2020.31
   221.2 2016.29   229.5 2015.92   241.5  2016.3   257.8 2018.48   279.2  2017.5
   283.3 2018.25   293.8  2024.4     304 2026.39   323.3 2027.07   345.4 2026.69
   386.7 2028.54     395 2029.52   411.6 2033.16   432.2 2032.46   440.5 2031.04
   448.8 2034.51   475.2 2039.27   538.5 2053.66   569.2 2061.61   607.2  2072.8
#Mann= 5 ,-1,0
       0      .1       0   221.2    .045       0   241.5      .1       0
  356.53     .06       0  456.53      .1       0
#XS Ineff= 2 , 0
                          277.96         2033.77
Permanent Ineff=
       F       F
Bank Sta=221.2,241.5
XS Rating Curve= 0 ,0
Exp/Cntr(USF)=0,0
Exp/Cntr=0.3,0.1

Type RM Length L Ch R = 1 ,7491    ,146.7,146.8,147.1
XS GIS Cut Line= 3
2187643.24880332630467.2777160732187625.74028995630588.670075484
2187823.00287399630973.857369768
#Sta/Elev= 30
       0 2086.27      10 2080.44      27 2072.87    62.5 2054.61    74.7 2049.51
    90.8 2039.86     107 2031.87   119.1 2021.02   127.8 2014.23   132.2 2011.24
   136.7 2009.41   136.7  2009.4   145.6 2008.28   160.5 2009.41   187.2 2016.97
   195.1 2018.28   204.1 2018.55   222.1 2016.37   244.6 2017.67   282.4 2017.22
   298.5 2018.91   329.8 2024.61   361.4 2029.14   383.9 2029.48   397.4  2033.5
     425  2039.1   455.8 2042.33   496.6 2053.31   522.9  2062.7   555.4 2072.43
#Mann= 5 ,-1,0
       0      .1       0   136.7    .045       0   160.5      .1       0
  272.65     .06       0  382.65      .1       0
Bank Sta=136.7,160.5
XS Rating Curve= 0 ,0
Exp/Cntr(USF)=0,0
Exp/Cntr=0.3,0.1

Type RM Length L Ch R = 1 ,7345    ,114.1,113.9,113.8
XS GIS Cut Line= 3
2187488.00665138630499.9602743762187482.17048026630628.356039137
2187680.60029853631032.219081023
#Sta/Elev= 30
       0 2079.05    13.2 2071.72    25.2 2066.89    53.3 2051.08    65.3 2046.36
   105.3 2025.83   136.6 2013.52   151.7 2012.69   166.5 2007.18   178.4 2006.63
   190.4 2007.22   196.3 2008.17   205.2 2008.17   214.1 2010.27   226.3 2010.59
   241.2 2013.41   324.9 2012.54   348.8 2017.17   374.6 2020.84   393.6 2025.52
   420.5 2026.43   429.5 2029.97   438.4  2035.9   444.4 2037.72   459.2 2038.74
   481.5 2038.53   490.4 2039.73   526.1 2050.91     564 2064.65   578.5 2068.31
#Mann= 5 ,-1,0
       0      .1       0   166.5    .045       0   190.4      .1       0
  348.53     .06       0  508.53      .1       0
Bank Sta=166.5,190.4
XS Rating Curve= 0 ,0
Exp/Cntr(USF)=0,0
Exp/Cntr=0.3,0.1

Type RM Length L Ch R = 1 ,7231    ,108.7,109,108.5
XS GIS Cut Line= 3
2187368.88913349630542.460230981 2187367.6640917630655.164075682
2187559.99565277631037.377114235
#Sta/Elev= 30
       0 2056.54    14.7 2049.05    22.7 2046.79    38.7 2037.52    46.7 2034.67
    66.7 2024.88    82.7  2018.6   119.4 2006.89   156.3 2006.52   168.2 2007.38
   182.42005.486   193.9 2004.27   203.82005.459     218 2007.12   229.5 2006.38
   257.6  2008.1   281.4 2007.56   309.6 2009.78   352.3  2008.2   388.1 2021.19
   416.4 2027.73   437.4 2028.55   448.2 2034.69   464.2 2039.98   468.7 2040.81
     478 2039.62   486.6 2040.27   504.5 2049.63   513.5 2047.56   540.6 2057.31
#Mann= 5 ,-1,0
       0      .1       0   182.4    .045       0   203.8      .1       0
  412.71     .06       0  522.71      .1       0
#XS Ineff= 2 , 0
          142.08 2015.83  231.69         2016.78
Permanent Ineff=
       F       F
Bank Sta=182.4,203.8
XS Rating Curve= 0 ,0
Exp/Cntr(USF)=0,0
Exp/Cntr=0.3,0.1

Type RM Length L Ch R = 1 ,7122    ,171.8,173.7,171.3
XS GIS Cut Line= 4
2187242.88746411630579.3322016832187272.99324078630710.478170773
 2187355.4136738630864.646221812 2187480.8876309631091.381408219
#Sta/Elev= 30
       0 2068.03    30.6 2058.38    59.3 2045.63    71.7 2038.31    96.1 2026.12
   129.5 2010.97   150.7 2003.47   164.8 2003.15   191.9 2005.34   198.92003.503
   209.8 2002.58   218.92003.617   248.3 2004.83     263 2003.27   278.2 2006.47
     328 2005.98   364.8 2001.56     381 2004.02   387.7 2007.21   396.8 2014.21
   401.4 2016.71   415.1 2021.27   433.9 2026.11   457.5 2027.11   469.2 2031.99
     502 2040.84   516.3 2047.81   522.2 2049.17   543.1 2049.98   568.5 2058.31
#Mann= 4 ,-1,0
       0      .1       0   198.9    .045       0   218.9      .1       0
  489.37     .06       0
#XS Ineff= 2 , 0
                          336.61         2012.67
Permanent Ineff=
       F       F
Bank Sta=198.9,218.9
XS Rating Curve= 0 ,0
Exp/Cntr(USF)=0,0
Exp/Cntr=0.3,0.1

Type RM Length L Ch R = 1 ,6948    ,327.3,327.3,323.1
XS GIS Cut Line= 3
2187192.69639243630586.3356070342187181.02405018630767.256911925
2187352.60748127631174.621656485
#Sta/Elev= 30
       0 2063.11      87 2038.05   151.2 2017.41   163.2 2010.58   175.2 2007.18
   192.1 1999.15   200.7 1998.21   240.9 1999.61   257.2  2001.9   278.9 2001.41
   295.1 2003.84   322.3 2002.57   335.3 2000.62     347 2001.16   353.1 2000.36
   364.6 1999.53   370.52000.397   377.6 2003.16   387.4 2003.16   430.8 1997.64
   436.7 1998.21   443.8 2001.32   469.8 2021.72   482.9 2023.26   491.5 2022.83
   504.6 2032.21   526.3 2038.22     535 2038.84   582.7 2051.02   623.3 2063.54
#Mann= 5 ,-1,0
       0      .1       0   353.1    .045       0   370.5      .1       0
   461.3     .06       0   561.3      .1       0
#XS Ineff= 2 , 0
                          399.28         2008.62
Permanent Ineff=
       F       F
Bank Sta=353.1,370.5
XS Rating Curve= 0 ,0
Exp/Cntr(USF)=0,0
Exp/Cntr=0.3,0.1

Type RM Length L Ch R = 1 ,6621    ,205,207.5,210.2
XS GIS Cut Line= 3
2187143.67255498630598.0079492852187003.60444797630823.284154729
2187181.02405018631248.157412667
#Sta/Elev= 30
       0 2051.66      60 2037.55   126.2 2024.87   149.7 2019.31   190.7 2012.56
   219.8 2009.95   228.5 2008.03   253.4 2006.45   265.3 2004.16   271.7 2001.37
   282.4 1993.35     289 1992.12   303.8  1993.3     315 1994.93   349.8 1994.31
   380.9 1995.91   468.7 1996.79   510.1 1997.12   518.7 1995.27   536.1 1995.49
   545.4 2000.61   557.7 2010.59   560.7 2011.74   579.1 2012.89   583.8  2016.9
   588.1 2018.79   627.1 2025.13   676.9 2040.85   701.4 2046.94   725.7 2055.11
#Mann= 7 ,-1,0
       0      .1       0  265.27     .05       0   282.4    .045       0
   303.8     .05       0  405.27      .1       0  475.27     .06       0
  585.27      .1       0
#XS Ineff= 2 , 0
                          410.93         2004.04
Permanent Ineff=
       F       F
Bank Sta=282.4,303.8
XS Rating Curve= 0 ,0
Exp/Cntr(USF)=0,0
Exp/Cntr=0.3,0.1

Type RM Length L Ch R = 1 ,6413    ,44.1,44.1,44.5
BEGIN DESCRIPTION:
Structure XS 3
END DESCRIPTION:
XS GIS Cut Line= 6
2186913.78807188630585.8642233492186813.62759806630718.581298782
2186818.96474587 630932.067211012186875.89432246631109.972137865
2186925.76741042631229.639000539 2186998.2700669631338.579085778
#Sta/Elev= 30
       0 2040.78    14.7 2036.12    59.8 2026.66   120.2 2010.57   200.9 1995.43
   252.9 1994.26   260.9 1994.97   276.9 1993.74   288.9 1993.82   312.9 1989.77
     341  1989.6     3511987.613   357.1 1986.39   365.51987.603   369.1 1990.08
   373.1 1991.32   404.5 1989.79   490.2 1989.06   553.8 1990.97   583.3 1988.55
   600.7  1989.1   612.4 1992.15     631 1994.62     644 2002.06     657 2007.26
   678.7 2007.78   687.3  2013.1   691.7 2014.43   784.5 2035.54   827.4 2049.26
#Mann= 9 ,-1,0
       0      .1       0   89.02     .06       0     351    .045       0
   365.5     .06       0  375.79     .08       0  474.53      .1       0
  514.53     .08       0  576.86     .06       0  756.51      .1       0
#XS Ineff= 2 , 0
                          555.96         1996.17
Permanent Ineff=
       F       F
Bank Sta=351,365.5
XS Rating Curve= 0 ,0
Exp/Cntr(USF)=0,0
Exp/Cntr=0.3,0.1

Type RM Length L Ch R = 1 ,6369    ,277,272.2,266
BEGIN DESCRIPTION:
Structure XS 2
END DESCRIPTION:
XS GIS Cut Line= 6
2186869.81518414630588.0834396742186769.65471032630720.800515108
2186774.99185813630934.2864273352186831.92143472 631112.19135419
2186881.79452268631231.8582168642186966.77336928631358.945487739
#Sta/Elev= 30
       0 2032.34    80.3 2012.67    87.1 2010.21   100.7 2001.43   107.5 1999.13
   172.2 1993.47   186.7 1993.01   214.7  1994.2   246.7 1991.64   266.7 1991.94
   286.7 1989.97   334.8 1989.95   354.3 1986.71   358.9 1985.97     3731986.666
   383.1 1988.73   542.6 1987.45   585.3 1989.85   593.9 1987.65   620.2 1990.12
   635.1 1990.39   645.9 1993.77   658.9 2000.66   680.6 2007.79   702.9  2009.3
   716.5 2015.15   779.9 2028.93   813.6 2038.23   832.8 2045.15   849.4 2049.05
#Mann= 7 ,-1,0
       0      .1       0      20     .06       0   354.3    .045       0
     373     .08       0  474.53      .1       0  646.86     .06       0
  796.51      .1       0
#XS Ineff= 2 , 0
                          583.39          1994.6
Permanent Ineff=
       F       F
Bank Sta=354.3,373
XS Rating Curve= 0 ,0
Exp/Cntr(USF)=0,0
Exp/Cntr=0.3,0.1

Type RM Length L Ch R = 1 ,6097    ,264,259.2,252.7
BEGIN DESCRIPTION:
Structure XS 1
END DESCRIPTION:
XS GIS Cut Line= 3
 2186372.1707608630932.4934068442186513.07146287630954.909427628
 2186882.9358058631406.432131988
#Sta/Elev= 30
       0 2054.29    12.2  2049.4    28.4 2039.45    40.5 2036.92    68.9 2021.88
   101.3 2007.37   109.4 2005.22   129.6 1993.64   146.5  1985.7   160.2 1982.94
   181.8 1983.49   188.71982.074   200.5 1981.67   206.2 1981.99     217 1983.85
   300.7 1982.14   388.1 1982.25   450.6 1985.44   471.4 1984.43   486.9 1985.94
   493.3 1987.25   502.4 1993.33   521.7 2000.81   551.6 2003.68     570 2007.91
   581.4 2008.38   585.1 2009.73   590.3 2014.52   595.7 2016.25   726.3 2041.47
#Mann= 5 ,-1,0
       0      .1       0   188.7    .045       0   206.2      .1       0
  542.67     .06       0  692.67      .1       0
#XS Ineff= 2 , 0
                          431.33         1997.94
Permanent Ineff=
       F       F
Bank Sta=188.7,206.2
XS Rating Curve= 0 ,0
Exp/Cntr(USF)=0,0
Exp/Cntr=0.3,0.1

Type RM Length L Ch R = 1 ,5838    ,82.3,83.8,85.9
XS GIS Cut Line= 3
  2186284.107822631156.653614682 2186641.1630102631270.334862943
2186833.30033121631443.258451847
#Sta/Elev= 30
       0  2029.3     4.3 2027.93    14.9 2022.14      63 2007.17    88.2 1999.92
   124.7 1991.48   138.6 1980.48   153.81977.362   180.6 1977.32     189 1978.31
   222.6 1976.69   236.1 1979.46   281.3 1980.76   310.7 1978.81   318.2 1979.36
   327.5  1981.8   350.7 1980.98   370.9  1982.6     376 1983.81   384.9 1988.79
   390.9 1990.87   449.7 1999.45   459.5 2001.58   470.3 2005.51   497.2  2006.5
   504.5 2010.55   526.1 2016.76   545.6  2019.7   613.9 2036.29   633.2 2038.93
#Mann= 5 ,-1,0
       0      .1       0   153.8    .045       0   180.6      .1       0
  444.72     .06       0  584.72      .1       0
Bank Sta=153.8,180.6
XS Rating Curve= 0 ,0
Exp/Cntr(USF)=0,0
Exp/Cntr=0.3,0.1

Type RM Length L Ch R = 1 ,5754    ,119,117.4,116.2
XS GIS Cut Line= 3
2186268.80160586631216.2332156092186507.68475496631331.387143891
2186756.36823838 631429.39048711
#Sta/Elev= 30
       0 2029.65    18.2 2020.53    52.6 2006.23    74.8 1998.86   105.1 1990.72
   123.6 1979.32   128.1 1978.29     137 1977.61   146.91975.071     153 1975.01
   163.6 1975.27   170.41976.724   190.2 1977.83   216.9 1976.06   221.3 1976.57
   227.9  1978.5     304 1979.56   321.6 1980.53   343.1 1986.12   357.4 1987.62
   373.2 1991.34   418.1 1998.59   436.6 2003.55   463.5 2004.53   467.4 2006.33
   472.1 2009.91   476.4 2011.72   485.9 2014.15   497.9 2015.88   532.5 2024.36
#Mann= 4 ,-1,0
       0      .1       0   146.9    .045       0   170.4      .1       0
  435.19     .06       0
Bank Sta=146.9,170.4
XS Rating Curve= 0 ,0
Exp/Cntr(USF)=0,0
Exp/Cntr=0.3,0.1

Type RM Length L Ch R = 1 ,5636    ,110.1,113.8,116.3
BEGIN DESCRIPTION:
Disconnected without IFA
END DESCRIPTION:
XS GIS Cut Line= 2
2186215.25861531631345.5886470042186761.24883583631518.512235908
#Sta/Elev= 30
       0 2039.66    13.5 2031.12    89.1  1995.7    97.5 1989.57   105.6 1982.06
   110.1 1976.43   111.9 1975.43   115.1 1974.51   131.1 1975.09   147.8  1973.9
   156.2 1973.72   166.1 1973.97   185.2 1976.57   210.8 1976.56   227.5 1974.39
   255.3 1977.26   328.2 1976.66   336.6 1978.91   349.2 1984.07     370 1987.96
   416.3 1997.04   445.7 1998.37   454.1 2003.81   466.7 2007.84   491.9 2014.94
   503.9  2017.1   529.6  2025.7   558.1 2030.66   564.4 2034.52   572.7 2037.29
#Mann= 5 ,-1,0
       0      .1       0   147.8    .045       0   166.1      .1       0
     370     .06       0     550      .1       0
#XS Ineff= 2 , 0
                          304.92         1985.33
Permanent Ineff=
       F       F
Bank Sta=147.8,166.1
XS Rating Curve= 0 ,0
Exp/Cntr(USF)=0,0
Exp/Cntr=0.3,0.1

Type RM Length L Ch R = 1 ,5523    ,184.4,179,174
BEGIN DESCRIPTION:
Disconnected without IFA
END DESCRIPTION:
XS GIS Cut Line= 3
2186197.64602755631406.4321319882186493.85773076631628.991195485
2186657.17445362631677.025525736
#Sta/Elev= 30
       0 2035.45     8.2 2031.91    20.9 2024.77    35.2 2017.86    51.2 2011.95
    78.2 2000.06    97.8 1987.93   113.2 1973.47   123.2 1972.25   132.3 1973.27
   136.31972.327   143.8 1971.61   154.6 1972.37   163.3 1974.32   192.3 1975.01
     258 1974.28   278.3 1973.01   289.4 1973.33   298.4 1972.01   308.4 1972.82
   318.4 1976.58   333.4 1986.19     338 1987.08   368.4  1988.9   393.8 1997.93
   402.1 1999.33     448 2011.14   456.3  2012.5   489.7 2021.88   540.7 2034.64
#Mann= 5 ,-1,0
       0      .1       0   136.3    .045       0   154.6      .1       0
     220     .06       0   450.5      .1       0
#XS Ineff= 2 , 0
                          309.29         1985.15
Permanent Ineff=
       F       F
Bank Sta=136.3,154.6
XS Rating Curve= 0 ,0
Exp/Cntr(USF)=0,0
Exp/Cntr=0.3,0.1

Type RM Length L Ch R = 1 ,5344    ,199.4,190,178
BEGIN DESCRIPTION:
Structure XS 4
END DESCRIPTION:
XS GIS Cut Line= 4
 2186111.1842331631476.8824830232186229.60026857631658.473301883
  2186407.868773631674.7797444192186634.18886201631724.694587428
#Sta/Elev= 30
       0 2041.97    38.6 2029.15    58.7 2020.24   105.4 1996.96   148.3 1979.91
     157 1978.39   162.9 1975.75   168.6 1974.35   227.4 1972.82   235.4 1969.96
   243.81968.951   255.5 1967.86     2641968.967   299.7    1973   347.9 1972.19
     368 1970.19   375.8 1970.76   379.9 1972.26   396.1 1981.97   424.9 1984.45
   445.1 1984.22   453.5 1988.67   469.8 1991.48   482.4 1995.28   502.6 2002.88
   531.3 2010.17   550.7 2016.29     560 2017.98   596.8 2029.62   627.6 2037.67
#Mann= 5 ,-1,0
       0      .1       0   243.8    .045       0     264      .1       0
  356.79     .06       0   565.8      .1       0
#XS Ineff= 2 , 0
          225.68 1980.42  416.97         1980.79
Permanent Ineff=
       F       F
Bank Sta=243.8,264
XS Rating Curve= 0 ,0
Exp/Cntr(USF)=0,0
Exp/Cntr=0.3,0.1

Type RM Length L Ch R = 1 ,5154    ,63.4,62.6,62.8
BEGIN DESCRIPTION:
Structure XS 3
END DESCRIPTION:
XS GIS Cut Line= 6
2185815.18376502632095.0846980452186052.08890768632004.817348254
2186261.02270575631900.3349107012186290.10498179631871.367935095
2186382.91820723631788.3390301862186592.95186323631831.313203194
#Sta/Elev= 30
       0 2013.32    18.2 2008.13      31 2006.01    43.9 2001.85      61 1998.38
    95.2 1988.62   132.4 1985.92     151 1981.38   162.6 1979.66   202.2 1979.65
   227.9 1977.16   250.2 1971.43   285.1 1970.02   294.9  1970.9   351.4 1971.66
   455.1 1967.79   553.9 1970.46   573.7 1967.29   579.4 1965.25   603.4 1965.52
   609.4 1967.24   616.9 1968.85   674.5 1971.65   691.3 1985.45   714.8 1990.11
   744.1 1998.41   779.4 2010.15   788.9 2011.65   821.5 2021.07   867.1 2036.05
#Mann= 7 ,-1,0
       0      .1       0     170     .06       0  487.14      .1       0
   573.7    .045       0   609.4      .1       0  632.05     .06       0
  743.47      .1       0
#XS Ineff= 2 , 0
          431.69 1976.25
Permanent Ineff=
       F       F
Bank Sta=573.7,609.4
XS Rating Curve= 0 ,0
Exp/Cntr(USF)=0,0
Exp/Cntr=0.3,0.1

Type RM Length L Ch R = 1 ,5091    ,155.2,165.9,176.5
BEGIN DESCRIPTION:
Structure XS 2
END DESCRIPTION:
XS GIS Cut Line= 6
 2185823.9027414632137.5683014282186090.14595664632034.699592785
2186307.05286182631942.5085950332186337.47460432631916.890285566
2186409.52609969631843.2376458472186588.75202722 631872.14742107
#Sta/Elev= 30
       0 2012.93    38.9  2002.5    80.9 1994.99     118 1992.17   163.2 1986.77
   240.4 1970.91   274.7 1970.34   283.3 1968.97   297.3 1969.83   326.7 1969.17
   358.4 1969.91   376.8 1968.26   392.8 1968.59   413.4 1967.62   465.2 1966.95
   471.3 1968.07   577.3 1968.15   598.21966.018   616.2 1964.91   624.8 1965.96
   633.4 1967.45     639 1969.73   656.3 1979.69   703.2 1991.47   723.1 1998.59
   743.3 2004.39   755.9 2009.26   780.2 2015.91   836.8 2036.57   845.5 2040.33
#Mann= 6 ,-1,0
       0      .1       0     170     .06       0  580.89      .1       0
   598.2    .045       0   624.8     .06       0  723.92      .1       0
#XS Ineff= 2 , 0
           389.8 1979.53
Permanent Ineff=
       F       F
Bank Sta=598.2,624.8
XS Rating Curve= 0 ,0
Exp/Cntr(USF)=0,0
Exp/Cntr=0.3,0.1

Type RM Length L Ch R = 1 ,4925    ,263.1,271.7,276.5
BEGIN DESCRIPTION:
Structure XS 1
END DESCRIPTION:
XS GIS Cut Line= 3
2185827.78168462632144.5596735142186128.79682086632032.479569595
2186559.50464877632051.693301695
#Sta/Elev= 30
       0 2011.91    21.8 2006.27    51.6 2001.66    77.2 1995.91   149.8 1988.67
   192.5 1982.92   222.4 1972.79   230.9 1971.56   260.8 1970.44   273.6 1968.16
   286.4 1969.38   352.6 1968.47   394.1 1965.68   444.7 1967.11   452.7 1966.07
   463.1 1968.04   536.8  1964.5   560.8 1966.45   567.1 1964.76   578.1 1963.41
   591.71964.795   604.9 1971.38   628.9 1988.88   656.9 2001.13   668.9 2008.23
   680.9 2017.34     693 2024.16     705 2027.69     721 2036.36   752.3  2045.9
#Mann= 5 ,-1,0
       0      .1       0     160     .06       0   371.2      .1       0
   567.1    .045       0   591.7      .1       0
#XS Ineff= 2 , 0
          373.04 1980.05
Permanent Ineff=
       F       F
Bank Sta=567.1,591.7
XS Rating Curve= 0 ,0
Exp/Cntr(USF)=0,0
Exp/Cntr=0.3,0.1

Type RM Length L Ch R = 1 ,4653    ,315.9,311.8,304.4
XS GIS Cut Line= 4
2185867.81029316632259.8420661172186083.96477929632157.368828248
2186282.50667766632298.2695303182186465.03713261632295.067241634
#Sta/Elev= 30
       0 2009.95    40.2 2002.95    53.5 1999.69    71.6 1997.06    93.4 1991.86
   159.8 1984.23   164.2 1983.48     173  1979.7     204 1978.58   226.2 1972.45
     245  1965.4   342.6 1964.62   365.5 1962.61   437.2 1960.01   445.5 1958.81
   451.5 1960.03   474.5 1968.59   488.3  1978.3   520.3 1992.39   548.3 2002.98
   556.4 2004.51   572.4 2005.37   576.4 2006.28   588.4 2011.79   596.4 2012.27
   600.4  2013.5   624.4 2025.82   640.4 2027.69   652.4 2035.45   665.2 2041.49
#Mann= 5 ,-1,0
       0      .1       0     120     .06       0     230      .1       0
   437.2    .045       0   451.5      .1       0
Bank Sta=437.2,451.5
XS Rating Curve= 0 ,0
Exp/Cntr(USF)=0,0
Exp/Cntr=0.3,0.1

Type RM Length L Ch R = 1 ,4342    ,385.7,387.3,387.3
XS GIS Cut Line= 4
2185880.61944789632552.8514806482186063.14990285632557.654913674
2186287.31011068632516.0251607892186442.62111183632448.777098438
#Sta/Elev= 30
       0 2018.95    31.6 2008.89    51.6  2006.4    55.6  2004.6    59.6 2001.03
    63.6 1999.99   119.6 1995.61   130.7 1992.81   147.6 1984.52   175.6 1982.81
   183.9 1978.71     208 1958.66   223.2 1956.94   232.5  1956.4   237.71956.893
     265  1959.3   355.4 1958.51   395.2 1963.14   410.6 1963.14   422.2 1966.63
   446.9 1977.04   463.8 1987.11   476.9 1990.89   491.3 2001.02   503.1 2006.67
   513.8 2013.61     529 2016.97   537.9 2022.61   556.4  2030.9   579.8 2039.24
#Mann= 5 ,-1,0
       0      .1       0     100     .06       0  192.59      .1       0
   223.2    .045       0   237.7      .1       0
Bank Sta=223.2,237.7
XS Rating Curve= 0 ,0
Exp/Cntr(USF)=0,0
Exp/Cntr=0.3,0.1

Type RM Length L Ch R = 1 ,3954    ,313.3,310.9,306.7
XS GIS Cut Line= 2
2185863.00686013632908.3055245072186473.04285432632874.681493331
#Sta/Elev= 30
       0 2018.55    74.2  1990.8    85.3 1987.73    89.3 1985.33    97.3 1977.65
   121.4 1976.89   141.4 1968.89   177.4 1961.87   225.5 1961.41   269.9 1963.25
   301.6 1954.92   330.6  1955.8   345.7 1954.09   393.8 1953.98   401.8 1952.65
   413.4 1951.25   417.11952.612   433.8 1965.51   453.9 1976.81   465.9 1986.83
   477.9 1992.97   489.9 2002.12   493.9 2003.71   510.9    2005     526 2018.34
     530 2020.69   582.1 2048.28   594.1 2051.47   606.1 2060.13     611 2061.94
#Mann= 5 ,-1,0
       0      .1       0      20     .06       0     120      .1       0
   401.8    .045       0   417.1      .1       0
Bank Sta=401.8,417.1
XS Rating Curve= 0 ,0
Exp/Cntr(USF)=0,0
Exp/Cntr=0.3,0.1

Type RM Length L Ch R = 1 ,3643    ,258.9,257.7,252.1
XS GIS Cut Line= 4
2185841.99167506633232.0099413682186113.52425787633179.970763296
 2186306.4548655633168.0185738952186495.65785908633135.462413829
#Sta/Elev= 30
       0    2038    63.3 2017.48    95.9 2007.84   120.3 2002.17   185.5 1981.51
   212.8 1971.68   226.2 1962.44   234.4 1963.08   253.8 1962.03     271 1956.89
   293.4  1952.7   331.2  1953.5     342 1948.72   351.3  1947.6   375.3 1948.71
   419.4 1950.19   451.4  1953.9   459.5 1953.24   470.3 1956.43   508.4 1973.55
   528.3  1984.1   540.5 1986.66   556.8 1997.35   564.9 2003.81   577.6 2006.15
   605.5 2018.92   613.6 2023.96   625.8 2027.37   633.9 2032.48   661.8 2045.73
#Mann= 7 ,-1,0
       0      .1       0     240     .06       0  336.47      .1       0
     342    .045       0   375.3      .1       0  436.47     .12       0
  639.77      .1       0
Bank Sta=342,375.3
XS Rating Curve= 0 ,0
Exp/Cntr(USF)=0,0
Exp/Cntr=0.3,0.1

Type RM Length L Ch R = 1 ,3386    ,163.1,162.6,161.9
XS GIS Cut Line= 3
2185866.52990577633456.6233914912186153.18968468633438.247764637
2186378.59737409633321.868794565
#Sta/Elev= 30
       0 2041.24     5.7 2038.53    13.7 2036.04    25.7 2031.15    40.9 2026.51
      50 2023.04    93.8 2003.97   105.9 1999.31   139.4 1987.57     154 1981.62
     166  1977.7   203.6 1961.13   222.1 1953.56   230.1 1950.95   246.1 1948.19
   283.5 1949.71   295.1 1949.25   304.1 1947.84   334.8  1947.4   340.1 1946.78
     3461945.272   361.5 1944.39   364.31944.714   371.6 1946.45   394.1 1948.19
   447.6 1947.98   506.7 1949.39   533.7 1954.06   538.2 1955.55   540.9 1957.18
#Mann= 6 ,-1,0
       0      .1       0     210     .06       0     346    .045       0
   364.3     .06       0  417.25      .1       0  537.25     .12       0
#XS Ineff= 2 , 0
          285.25 1960.58
Permanent Ineff=
       F       F
Bank Sta=346,364.3
XS Rating Curve= 0 ,0
Exp/Cntr(USF)=0,0
Exp/Cntr=0.3,0.1

Type RM Length L Ch R = 1 ,3223    ,215.5,224.1,223.7
XS GIS Cut Line= 4
 2185900.8310759633581.5776540942186260.99336222633566.877152612
2186292.84444877633547.2764839682186530.50255607633483.574310876
#Sta/Elev= 30
       0  2033.9    86.5 1996.11   123.4 1981.49   135.5 1975.42   143.5 1968.18
   147.5  1965.9   151.5  1964.7   163.5 1963.83   167.5 1961.94   179.5 1953.83
   195.5 1946.94   211.5 1946.14   242.1 1946.75   287.6 1944.98   335.6  1946.2
   372.81943.661   381.5 1943.58   389.91943.958   442.7 1946.93     509 1945.71
   529.7 1955.27   562.8 1975.55   571.1 1976.74   579.4 1983.63     595 1992.22
   611.3 2004.41   624.4 2007.88   629.1 2010.78   637.4 2017.54   643.9 2020.96
#Mann= 5 ,-1,0
       0      .1       0     270     .06       0   372.8    .045       0
   389.9     .06       0  477.86      .1       0
#XS Ineff= 2 , 0
          325.14 1957.41
Permanent Ineff=
       F       F
Bank Sta=372.8,389.9
XS Rating Curve= 0 ,0
Exp/Cntr(USF)=0,0
Exp/Cntr=0.3,0.1

Type RM Length L Ch R = 1 ,2999    ,58.2,57.7,57.6
XS GIS Cut Line= 4
2185924.79601849633690.9965731762186257.31823685633700.406707747
2186483.53903761633710.4302445792186559.90355904633679.580997313
#Sta/Elev= 30
       0 2024.65    79.5 1990.47    87.4 1984.84    91.4 1982.98   103.4 1982.33
   131.4 1967.27   147.4 1957.36   151.4 1954.64   159.4 1947.07   163.4 1944.83
   186.5  1942.7   227.5 1942.39   339.5 1945.45   371.6 1942.22   391.6 1942.72
   419.6 1941.68   451.6 1943.29   471.6 1942.71   479.7 1943.73   487.7 1942.78
   493.8 1940.64   499.7 1939.19   508.7  1939.6   519.7 1940.38   531.7 1949.16
   539.7 1956.44   555.7 1965.41   573.1 1970.69   591.3 1980.88   641.5 2005.63
#Mann= 5 ,-1,0
       0      .1       0  352.66     .06       0  452.66      .1       0
   493.8    .045       0   508.7      .1       0
#XS Ineff= 2 , 0
          332.79 1959.26
Permanent Ineff=
       F       F
Bank Sta=493.8,508.7
XS Rating Curve= 0 ,0
Exp/Cntr(USF)=0,0
Exp/Cntr=0.3,0.1

Type RM Length L Ch R = 1 ,2941    ,116.3,117.9,118.8
XS GIS Cut Line= 5
2185896.05048649633767.2176985942185934.41294674633768.163371969
2186259.76832043 633765.333922632186441.01996749633764.917747319
2186577.11723653633692.866251942
#Sta/Elev= 30
       0 2043.44     4.1 2041.41    12.1  2035.3    24.1 2032.21    36.1 2024.64
    56.1 2015.43    76.1 2004.76   113.8  1988.2   120.1 1983.29   136.1 1981.92
   140.1 1979.93   148.1  1974.3   160.1 1967.62   192.1 1945.53   200.1 1942.08
   260.1 1941.48   340.1  1942.2   372.3 1943.62   392.1 1941.47   440.2 1940.53
   504.3 1942.93   513.51940.214   520.1 1938.79   527.91940.122   540.1 1943.78
   564.9 1956.01   604.3 1968.76   630.1 1982.13   671.4 1996.08     699 2010.58
#Mann= 5 ,-1,0
       0      .1       0  373.74     .06       0  473.74      .1       0
   513.5    .045       0   527.9      .1       0
#XS Ineff= 2 , 0
          364.66 1956.57
Permanent Ineff=
       F       F
Bank Sta=513.5,527.9
XS Rating Curve= 0 ,0
Exp/Cntr(USF)=0,0
Exp/Cntr=0.3,0.1

Type RM Length L Ch R = 1 ,2823    ,359.4,362.9,365.6
BEGIN DESCRIPTION:
Structure XS 4
END DESCRIPTION:
XS GIS Cut Line= 3
2185930.25492248 633822.558943622186458.63255525 633888.20586163
2186591.52753561633814.553221911
#Sta/Elev= 30
       0 2027.08       6 2022.72    26.1 2011.64    42.2 2005.49    78.5 1988.38
    86.6  1983.5   102.7 1982.24   118.9 1974.85     143 1958.87   151.1 1951.18
   161.8 1942.55   167.2 1940.81   206.3 1938.75   219.6 1940.27   231.7 1939.63
   292.1 1941.51   340.5  1941.8   348.6 1942.76   376.6 1940.92   466.6 1938.69
   477.6  1938.1   493.7 1938.77   505.8 1943.92   517.9 1942.03   525.9 1943.05
   547.9 1953.41   566.2 1960.48   621.1 1975.18   648.5 1983.76   684.4 1991.77
#Mann= 5 ,-1,0
       0      .1       0     350     .06       0     450      .1       0
   466.6    .045       0   493.7      .1       0
#XS Ineff= 2 , 0
          309.31 1954.97
Permanent Ineff=
       F       F
Bank Sta=466.6,493.7
XS Rating Curve= 0 ,0
Exp/Cntr(USF)=0,0
Exp/Cntr=0.3,0.1

Type RM Length L Ch R = 1 ,2460    ,131,131.4,131.4
BEGIN DESCRIPTION:
Structure XS 3
END DESCRIPTION:
XS GIS Cut Line= 6
2185941.81234938633959.9271357912186287.85452661633969.193078724
2186310.99086364634223.9355408822186360.64689896  634241.5070072
2186374.93780765634451.8578418332186558.96726672634439.103737524
#Sta/Elev= 30
       0  2024.2    17.6 2014.61    30.4 2012.64    54.2 1999.79    62.4 2000.28
   134.4 1975.59   157.4 1964.05   186.4  1946.2   206.4 1937.62   309.5  1939.2
   326.5 1937.66   394.6 1937.58   426.7 1936.04   450.8 1936.99   555.2 1933.37
   602.6 1932.96   611.21930.427   632.7 1928.74   640.11930.457   650.6  1936.5
   655.5 1937.09   747.4 1933.72   791.5 1930.04   855.5 1929.77   885.3 1928.32
   903.5 1929.17   918.8 1931.92   959.8 1932.07  1031.9 1960.41  1050.8 1969.74
#Mann= 9 ,-1,0
       0      .1       0     230     .06       0  356.17      .1       0
  547.21     .06       0   611.2    .045       0   640.1     .06       0
   685.3     .07       0   725.3      .1       0   965.6     .06       0
#XS Ineff= 2 , 0
                          673.22         1955.46
Permanent Ineff=
       F       F
Bank Sta=611.2,640.1
XS Rating Curve= 0 ,0
Exp/Cntr(USF)=0,0
Exp/Cntr=0.3,0.1

Type RM Length L Ch R = 1 ,2329    ,137.5,140.8,142.9
BEGIN DESCRIPTION:
Structure XS 2
END DESCRIPTION:
XS GIS Cut Line= 6
2185947.27285111634067.6755604552186250.76995978634063.431931859
2186284.11408874 634350.83932816 2186323.8583581634367.771786704
2186339.17004599634511.7525790532186555.30376678634487.407527019
#Sta/Elev= 30
       0  2029.6    12.9  2020.3    24.9 2018.95    44.9 2006.83    82.3 1989.91
    96.9 1986.38   124.9 1974.47   164.9 1962.79   176.9 1953.25   192.9 1947.15
   204.9 1939.12   208.9 1938.22   276.9 1934.73   303.5 1936.39   450.2  1934.1
   499.5  1930.8   587.4  1931.5     604 1928.18   625.4 1928.24   657.7 1932.45
   722.1 1927.73   786.1 1926.83   798.2 1928.77   862.6 1926.47     882 1930.61
   906.9 1929.59   914.9 1930.94   943.1 1946.55   979.7  1956.8   998.6 1964.08
#Mann= 10 ,-1,0
       0      .1       0     230     .06       0  408.88      .1       0
  427.45     .06       0  509.66     .07       0     604    .045       0
   625.4     .07       0  633.06     .06       0  811.08      .1       0
  911.08     .06       0
#XS Ineff= 2 , 0
          588.45 1940.48
Permanent Ineff=
       F       F
Bank Sta=604,625.4
XS Rating Curve= 0 ,0
Exp/Cntr(USF)=0,0
Exp/Cntr=0.3,0.1

Type RM Length L Ch R = 1 ,2188    ,189.2,186.5,184.9
BEGIN DESCRIPTION:
Structure XS 1
END DESCRIPTION:
XS GIS Cut Line= 4
 2185965.5096489634414.1839315532186128.82637175634399.773632478
2186468.26897219634644.7487167592186597.96166387  634607.9223969
#Sta/Elev= 30
       0 2008.18    14.5 2004.97    26.8 2000.66    50.9 1989.97    70.9 1978.77
      79 1975.41   107.1 1968.55   151.3 1938.03   164.5 1931.44   177.9 1929.83
   237.1 1929.45   253.3 1927.73   291.4  1929.2   299.2 1927.14   303.1 1925.93
   316.1 1925.43   323.6 1927.22   327.8  1929.5   336.4 1931.34   355.5 1928.97
   399.9  1929.1   410.9 1927.02   528.2  1926.2   557.8 1924.36   594.7 1929.65
   611.6 1935.72   661.5 1949.19   694.7 1962.12     703 1963.09   717.4 1969.75
#Mann= 5 ,-1,0
       0      .1       0   299.2    .045       0   323.6      .1       0
  343.95     .06       0  582.56      .1       0
#XS Ineff= 2 , 0
          237.52 1940.84
Permanent Ineff=
       F       F
Bank Sta=299.2,323.6
XS Rating Curve= 0 ,0
Exp/Cntr(USF)=0,0
Exp/Cntr=0.3,0.1

Type RM Length L Ch R = 1 ,2002    ,273.9,267.5,257.9
XS GIS Cut Line= 4
2185930.25492248634605.5185267132186085.56592363634611.923104079
2186407.39593631634768.8352495662186620.34813376634699.986042873
#Sta/Elev= 30
       0 2018.81    29.9 2003.59      42 1998.87      66 1985.34    74.6 1983.11
    97.6 1969.85   116.9 1961.72   128.4 1953.73     150 1932.62   158.3 1927.94
   180.6 1926.17   233.1  1926.4     2461924.561   251.8 1923.75   269.6 1924.64
   298.9 1927.28   319.9 1925.73   340.9 1925.91   354.2 1927.36   443.2 1926.97
   478.8 1923.81   514.3 1923.91   526.9 1922.55   596.4 1924.45   606.8 1926.62
   636.2  1925.5     653 1933.01   686.7 1942.03   729.9 1957.02   737.3 1958.38
#Mann= 8 ,-1,0
       0      .1       0     246    .045       0   269.6     .06       0
  365.44      .1       0  475.44     .06       0  495.44      .1       0
  553.49     .06       0  683.49      .1       0
#XS Ineff= 2 , 0
                          626.59         1940.84
Permanent Ineff=
       F       F
Bank Sta=246,269.6
XS Rating Curve= 0 ,0
Exp/Cntr(USF)=0,0
Exp/Cntr=0.3,0.1

Type RM Length L Ch R = 1 ,1734    ,244,243.1,243.9
XS GIS Cut Line= 3
2185870.06231342634789.1775004862186045.77088316634908.756943777
2186655.87008362634757.452342061
#Sta/Elev= 30
       0 2022.66     7.4 2017.76    70.6 1982.52   131.1 1954.19   176.7 1938.24
   191.3 1933.77   203.1 1931.52   212.5 1927.52   231.5 1923.04   243.9 1921.31
   252.1 1920.25     267 1921.24   285.1    1924   313.9 1923.88   326.3 1922.46
   346.9 1924.64   389.2 1924.05     442 1920.82     454 1922.38   471.7 1922.17
   482.9 1923.91   515.9 1926.22   541.1 1925.88   564.2  1924.2   573.6 1921.57
   705.4 1923.65   717.8    1927   742.5 1927.25   752.4 1931.98   841.1 1959.95
#Mann= 6 ,-1,0
       0      .1       0   243.9    .045       0     267      .1       0
  342.54     .06       0  442.54      .1       0  752.54     .06       0
Bank Sta=243.9,267
XS Rating Curve= 0 ,0
Exp/Cntr(USF)=0,0
Exp/Cntr=0.3,0.1

Type RM Length L Ch R = 1 ,1491    ,129.2,128.9,130.1
XS GIS Cut Line= 3
2185789.52921896634947.8032926072185948.15501108 635147.91583036
2186826.69785975635008.813212654
#Sta/Elev= 30
       0 1972.03    22.2 1968.75    39.9 1960.88    93.6 1943.11   134.5 1933.55
   182.2 1927.96   324.3 1920.81   338.31917.995   366.2 1918.03   409.3 1919.89
   453.6 1917.94     470 1920.07   530.8 1917.84   656.3  1919.5   672.5 1916.38
   688.7 1916.23   717.1  1919.7   737.3 1918.18   761.6 1919.93   818.3 1918.45
   891.2 1921.02   925.6 1919.77   951.9  1915.5   976.2 1913.97   996.5 1922.93
  1012.7 1927.35    1041 1938.48  1093.4  1945.7  1128.3 1953.48  1144.8 1954.52
#Mann= 8 ,-1,0
       0      .1       0     140     .05       0  285.36      .1       0
   338.3    .045       0   366.2      .1       0  385.36     .06       0
  485.36      .1       0  985.36     .06       0
Bank Sta=338.3,366.2
XS Rating Curve= 0 ,0
Exp/Cntr(USF)=0,0
Exp/Cntr=0.3,0.1

Type RM Length L Ch R = 1 ,1362    ,171,173.9,171.6
XS GIS Cut Line= 4
2185758.01694394634973.7038696942185898.14534733635274.596605087
2186692.39067198635199.9163678112186872.50249847635131.481174435
#Sta/Elev= 30
       0 1966.72    34.7 1953.79    74.4 1941.34    96.5 1936.94   184.7 1924.65
   281.2 1920.95   426.4 1920.08   450.5 1915.86   482.6 1916.87   500.61914.648
   506.7 1913.52   524.21914.689   530.8 1917.22   554.9 1916.17     567 1918.17
   621.5 1915.11   643.6 1916.09   696.2 1914.19   731.6 1916.53   852.2  1916.2
   872.3 1913.94   888.4 1916.36     949 1915.29  1065.2 1917.23  1077.2 1913.16
  1085.3 1912.46  1105.3  1913.7  1131.6 1924.69  1181.2 1933.06  1322.3 1952.48
#Mann= 10 ,-1,0
       0      .1       0     200     .05       0     310      .1       0
   500.6    .045       0   524.2     .06       0  611.92      .1       0
  911.92     .05       0 1001.92      .1       0 1209.67     .05       0
 1269.67     .06       0
Bank Sta=500.6,524.2
XS Rating Curve= 0 ,0
Exp/Cntr(USF)=0,0
Exp/Cntr=0.3,0.1

Type RM Length L Ch R = 1 ,1188    ,137.6,138.5,139.1
XS GIS Cut Line= 4
2185684.91438114634919.4345144352185908.85564492635420.868277742
2186690.03563885635323.6244000942186909.67135102 635226.00852802
#Sta/Elev= 30
       0 1989.38    19.4 1978.06    41.3 1976.34    63.2 1965.23    85.1 1957.75
   181.5 1931.49   255.1  1924.1   461.9 1918.58   479.4 1917.18   501.3 1911.33
   629.1 1911.41   648.6 1912.53   665.4 1916.24   682.81911.394   689.6 1910.07
   699.41911.174   709.6 1913.09   773.3 1914.88   838.7 1913.28   915.3 1914.89
    1008 1911.19  1056.4 1913.97    1137 1912.78  1225.5 1914.74  1290.2 1911.34
  1318.4 1911.87  1352.2 1922.12    1400 1926.97  1421.9 1932.64  1576.7 1949.03
#Mann= 10 ,-1,0
       0      .1       0     260     .05       0     470      .1       0
   682.8    .045       0   699.4      .1       0  719.17     .06       0
  819.17     .05       0 1219.17      .1       0 1416.38     .05       0
 1526.38     .06       0
#XS Ineff= 2 , 0
          664.48 1922.96
Permanent Ineff=
       F       F
Bank Sta=682.8,699.4
XS Rating Curve= 0 ,0
Exp/Cntr(USF)=0,0
Exp/Cntr=0.3,0.1

Type RM Length L Ch R = 1 ,1050    ,112.9,113.3,113.5
XS GIS Cut Line= 4
2185678.55572002634997.1152294132185901.23785788 635552.40455553
2186780.33032052635487.1309858192186940.16506081 635362.90283066
#Sta/Elev= 30
       0  1959.4    60.4 1939.51    90.6 1924.45   232.8 1924.02   366.4  1918.3
   400.9 1912.03   573.4 1912.06   586.2 1908.41   613.3 1907.47   625.3 1909.43
   653.4 1909.99   742.2 1910.48   757.91908.676   782.11908.685   789.7 1911.73
   809.8 1911.82   844.9 1909.56     899 1911.64  1078.2 1908.86  1094.6 1910.84
  1166.8 1909.45  1214.9 1911.33  1335.2 1911.48  1399.4 1908.37  1407.4 1909.47
  1432.9 1919.83  1447.5 1923.21  1560.9 1927.32  1596.1 1932.43  1682.2 1939.51
#Mann= 10 ,-1,0
       0      .1       0     170     .06       0     270     .05       0
     380      .1       0   757.9    .045       0   782.1      .1       0
  878.28     .06       0  968.28     .05       0 1368.28      .1       0
 1589.79     .05       0
#XS Ineff= 2 , 0
          655.74 1919.63
Permanent Ineff=
       F       F
Bank Sta=757.9,782.1
XS Rating Curve= 0 ,0
Exp/Cntr(USF)=0,0
Exp/Cntr=0.3,0.1

Type RM Length L Ch R = 1 ,937     ,249.4,245.5,238.8
XS GIS Cut Line= 4
2185644.29853578 635035.159968852185909.33076002635663.058693029
2186799.20830423635607.5442161882186989.73437765635436.228360697
#Sta/Elev= 30
       0 1949.83    92.3 1923.35   188.9 1925.02   310.5 1918.63   327.8 1915.09
   357.1 1912.52   503.7 1912.69   670.8  1909.3   753.9 1909.66   840.91906.769
   852.7 1906.41   872.91906.867     969 1909.69  1049.1 1907.59  1125.2 1910.41
  1153.3 1909.95  1169.3 1906.51  1185.4 1908.46  1261.5 1909.25  1321.6 1907.09
  1357.7 1909.13  1425.8 1909.35  1469.9 1906.99  1481.9  1908.8    1506 1917.66
  1628.2  1923.8  1698.2 1922.88  1711.5  1926.5  1751.1 1931.47  1829.4 1938.95
#Mann= 11 ,-1,0
       0      .1       0     130     .06       0     240      .1       0
   840.9    .045       0   872.9      .1       0  951.54     .06       0
 1051.54     .05       0 1441.54      .1       0 1541.54     .05       0
 1663.15      .1       0 1793.15     .05       0
#XS Ineff= 2 , 0
           779.6    1919
Permanent Ineff=
       F       F
Bank Sta=840.9,872.9
XS Rating Curve= 0 ,0
Exp/Cntr(USF)=0,0
Exp/Cntr=0.3,0.1

Type RM Length L Ch R = 1 ,691     ,271.3,279.3,280.3
XS GIS Cut Line= 4
2185858.76045175 636103.722463592186120.27996982635866.473449015
2186794.02943945635631.5071645242187007.27247918635462.714404591
#Sta/Elev= 30
       0 2022.68    42.4 1994.34    51.4 1991.43    66.7 1978.81    99.1 1946.88
   121.7 1918.73   130.2 1911.23   153.1 1910.26   180.1 1904.25   196.3 1908.41
   265.7  1908.4   295.5  1903.4   349.1 1906.36   429.2 1902.74   437.7 1902.12
   450.4 1902.71   458.9 1905.25     514 1903.94   543.6  1907.4   717.3 1904.57
   751.2 1908.05   784.3  1904.8   912.2 1908.71   929.1 1905.62   971.5 1909.22
  1009.6 1917.92  1138.2 1921.93  1196.9 1920.94  1237.7 1928.87  1338.6    1938
#Mann= 9 ,-1,0
       0      .1       0   429.2    .045       0   450.4      .1       0
   513.1     .06       0   623.1     .05       0   723.1      .1       0
  1033.1     .05       0 1156.65      .1       0 1276.65     .05       0
#XS Ineff= 2 , 0
          347.73 1919.79
Permanent Ineff=
       F       F
Bank Sta=429.2,450.4
XS Rating Curve= 0 ,0
Exp/Cntr(USF)=0,0
Exp/Cntr=0.3,0.1

Type RM Length L Ch R = 1 ,412     ,193.3,186,180.9
BEGIN DESCRIPTION:
County boundary Structure XS 4
END DESCRIPTION:
XS GIS Cut Line= 4
 2185915.9905326636173.8180058082186088.58811292636159.341319262
2186713.08896306635808.0595910572187050.65316724635533.049996173
#Sta/Elev= 30
       0 2008.31    32.3 1989.97    44.3 1985.53    84.5 1959.89   100.5 1954.15
   148.9  1929.3   181.9  1908.9   256.7 1902.94   277.3 1905.45   365.5 1903.97
   402.2 1906.76   466.5 1901.41   488.8 1904.84   539.9 1905.68   550.5  1901.4
   581.2 1900.56   590.91901.373   600.4 1904.65     618 1905.06   732.9 1903.35
   788.4 1907.48   800.1  1905.8   884.1 1907.16   928.1  1912.5  1046.3 1916.36
  1104.4 1921.72  1185.6 1922.43  1270.3  1929.3  1301.3 1928.06  1325.1    1930
#Mann= 9 ,-1,0
       0      .1       0   550.5    .045       0   590.9      .1       0
  959.72     .06       0  999.72     .05       0 1079.72     .06       0
 1159.72      .1       0 1209.72     .06       0 1309.72     .05       0
#XS Ineff= 2 , 0
          402.91 1916.46  785.43         1917.41
Permanent Ineff=
       F       F
Bank Sta=550.5,590.9
XS Rating Curve= 0 ,0
Exp/Cntr(USF)=0,0
Exp/Cntr=0.3,0.1

Type RM Length L Ch R = 1 ,226     ,55.3,58.1,59.8
BEGIN DESCRIPTION:
Structure XS 3
END DESCRIPTION:
XS GIS Cut Line= 6
2185967.08112923636337.5750328322186110.00949998636342.040911302
2186344.80558953636241.5433903842186452.36102907636187.765670613
2186745.57764401 635934.242134552187049.55174168635532.381842626
#Sta/Elev= 30
       0 1977.75    33.1 1967.36    89.9 1942.34   109.3 1930.98   137.2 1909.97
   141.2 1908.06   149.7 1906.19   236.7 1907.25     379 1905.34   555.1 1905.35
   565.6 1904.09   582.71900.163   591.3 1898.58   638.9 1898.99   644.2 1900.23
   659.4 1904.83     702 1903.12   832.4 1901.57   859.7  1903.8   962.8 1905.59
   968.9 1906.21   992.9 1912.53  1043.2 1915.98  1108.2 1917.24  1123.1  1916.2
  1131.6 1917.22  1142.7 1916.04  1165.9 1917.95  1297.3 1922.47  1410.2 1929.97
#Mann= 5 ,-1,0
       0      .1       0   582.7    .045       0   644.2      .1       0
   906.3     .06       0  1396.3     .05       0
#XS Ineff= 2 , 0
                           912.2         1920.37
Permanent Ineff=
       F       F
Bank Sta=582.7,644.2
XS Rating Curve= 0 ,0
Exp/Cntr(USF)=0,0
Exp/Cntr=0.3,0.1

Type RM Length L Ch R = 1 ,168     ,151.8,159.8,169.5
BEGIN DESCRIPTION:
Structure XS 2
END DESCRIPTION:
XS GIS Cut Line= 6
2185957.15186037636402.4893494872186118.97245328 636400.94031867
2186373.28897765636288.5318004492186480.84441719636234.754080678
2186774.06103213635981.2305446152187078.03512979635579.370252691
#Sta/Elev= 30
       0 1974.64    94.6 1937.67     123 1928.27     155 1909.28   163.1 1906.33
   176.3 1904.99   237.5 1904.81   272.5 1906.94   316.2 1904.05   417.3 1903.58
   483.3 1905.97   514.7 1904.41     592 1904.83   606.2 1904.03   622.1  1899.7
   653.6 1898.04   669.3 1899.83   677.1 1903.44     685  1904.5     870 1901.05
   962.9 1903.71     993 1908.18    1013 1908.26  1030.8 1911.67  1123.7 1916.79
    1190 1919.22  1203.6 1918.23  1214.9 1920.48  1359.1 1925.47  1451.7 1930.61
#Mann= 7 ,-1,0
       0      .1       0   622.1    .045       0   669.3      .1       0
 1007.78     .06       0 1097.78     .05       0 1127.78     .06       0
 1417.78     .05       0
#XS Ineff= 2 , 0
          489.82 1918.28  955.92         1913.77
Permanent Ineff=
       F       F
Bank Sta=622.1,669.3
XS Rating Curve= 0 ,0
Exp/Cntr(USF)=0,0
Exp/Cntr=0.3,0.1

Type RM Length L Ch R = 1 ,8       ,,,
BEGIN DESCRIPTION:
Structure XS 1
END DESCRIPTION:
XS GIS Cut Line= 6
2186010.13659184636527.7020867022186168.90890735636527.702086702
2186729.14354595636268.071517794 2186890.2997139636171.584310281
2186994.10576604 635931.309741542187155.44217835635590.353446343
#Sta/Elev= 30
       0 1937.27      46  1920.5      78 1918.88     142 1906.16   166.8 1903.24
   237.3 1904.68   259.4 1903.01     396 1902.63     471 1899.94   602.4 1901.69
   629.7 1900.79   636.91899.022   678.5    1898   710.4 1898.86   735.4 1902.06
   748.7 1900.69     762 1902.14   805.2 1902.61   831.1 1898.19   906.5 1899.13
   929.8 1902.42  1010.3 1904.43  1183.4 1905.22  1223.8  1906.6  1245.9 1903.91
    1265 1906.21  1285.7 1914.17    1299 1916.55  1440.6 1922.07    1603 1930.51
#Mann= 5 ,-1,0
       0      .1       0   636.9    .045       0   710.4      .1       0
 1335.82     .06       0 1545.82     .05       0
#XS Ineff= 2 , 0
          402.02 1920.79
Permanent Ineff=
       F       F
Bank Sta=636.9,710.4
XS Rating Curve= 0 ,0
Exp/Cntr(USF)=0,0
Exp/Cntr=0.3,0.1
LCMann Table=0

Chan Stop Cuts=-1
Use User Specified Reach Order=0
Composite Channel Slope=5
